--- PNTRSRN.prj (project) ---

Proj Title=PNTRSRN
Current Plan=p01
Default Exp/Contr=0,0
English Units
Geom File=g01
Flow File=f01
Plan File=p01
BEGIN DESCRIPTION:
END DESCRIPTION:
DSS Export Rating Curves= 0
DSS Export Rating Curve Sorted= 0
DSS Export Volume Flow Curves= 0
DXF Filename=..\..\..\..\..\Engineering\Hydraulics\PNTRSRN\PNTRSRN.
DXF OffsetX= 0
DXF OffsetY= 0
DXF ScaleX= 0
DXF ScaleY= 0

--- PNTRSRN.p01 (plan) ---

Plan Title=Floodplain
Program Version=4.00
Geom File=g01
Flow File=f01
K Sum by GR=0
Std Step Tol=0.01
Critical Tol=0.01
Num of Std Step Trials=20
Max Error Tol=0.3
Flow Tol Ratio=0.001
Split Flow NTrial=30
Split Flow Tol=0.02
Split Flow Ratio=0.02
Log Output Level=0
Friction Slope Method=1
Unsteady Friction Slope Method=2
Unsteady Bridges Friction Slope Method=1
Global Log Level=0
CheckData=False
Run HTab=0
Run UNet=0
Run PostProcess=0
UNET Theta=0
UNET Theta Warmup=0
UNET ZTol=0
UNET ZSATol=0
UNET MxIter=0
UNET MaxInSteps=0
UNET DtIC=0
UNET DtMin=0
UNET MaxCRTS=0
UNET WFStab=0
UNET SFStab=0
UNET WFX=0
UNET SFX=0
UNET DSS MLevel=0
UNET DZMax Abort=0
UNET Convert EG Bridges=0
UNET Use Existing IB Tables=0
UNET Froude Limit=0
UNET Froude Power=0
Write IC File=0
Echo Input=False
Echo Output=False
Write Detailed=0

--- PNTRSRN.f01 (steady flow) ---

Flow Title=NFF Regression Equation
Program Version=4.10
Number of Profiles= 1
Profile Names=P100yr
River Rch & RM=PNTRSRN,Main            ,9518
881.7515
River Rch & RM=PNTRSRN,Main            ,8426.9
 950.767
River Rch & RM=PNTRSRN,Main            ,4041.9
1055.406
River Rch & RM=PNTRSRN,Main            ,650
1171.506
Boundary for River Rch & Prof#=PNTRSRN,Main            , 1
Up Type= 0
Dn Type= 3
Dn Slope=0.006
DSS Import GetInterval= 0
DSS Import GetPeak= 0
DSS Import FillOption= 0

--- PNTRSRN.g01 (geometry) ---

Geom Title=2003 WVU SAMB 3 Meter DEM
Program Version=4.10

River Reach=PNTRSRN         ,Main
Reach XY= 30
     1666490.782      647627.955     1666096.332      647194.637
     1665730.582      646958.164     1665612.825      646556.617
     1665653.896      646243.527     1665525.151      645938.561
     1665190.788      645532.589     1665150.858      645259.586
     1665006.326      645210.541     1665079.538      645061.617
     1665067.686      644929.012     1664751.737      644629.696
     1664435.741       644635.61     1663975.672      644337.867
     1663809.873      644119.985     1663809.873      643777.971
     1663593.835      643487.183     1663524.173      643238.702
     1663374.977      642961.999     1663092.709      642698.219
     1663009.029      642535.314     1662529.631      642493.257
     1662185.143      642802.828     1661847.817      642995.276
      1661731.15      642858.123     1661713.519      642679.881
     1661512.013       642638.15     1661469.056      642752.704
     1661281.227      642492.381       1661166.8      642449.274

Type RM Length L Ch R = 1 ,9518    ,172.7,173.2,173.4
XS GIS Cut Line= 2
     1666541.615      647563.973     1666368.004      647725.649
#Sta/Elev= 28
       0  859.24     9.5  856.35      19  853.46    28.5  850.66      38  847.89
    47.4  845.14    56.9  841.78    66.4  837.61      75   834.5    75.9  834.18
    85.4  833.38      90  833.83    94.9   834.3   104.4  835.34   113.9  835.92
   123.4  836.44   132.8  837.11   142.3   838.1   151.8  839.07   161.3  840.22
   170.8   841.9   180.3  844.02   189.8  846.56   199.3  849.05   208.8  851.47
   218.2  853.74   227.7  856.03   237.2  858.61
#Mann= 3 , 0 , 0
       0      .1       0    75.9    .045       0    94.9      .1       0
Bank Sta=75.9,94.9
XS Rating Curve= 0 ,0
Exp/Cntr=0.3,0.1

Type RM Length L Ch R = 1 ,9344.8  ,138.5,139.4,140.1
XS GIS Cut Line= 2
     1666422.257      647441.361     1666256.242        647591.1
#Sta/Elev= 26
       0  855.63     9.7  853.32    19.4  850.91    29.2  848.37    38.9  845.54
    48.6  842.61    58.3  839.53      68  836.01    77.8  832.68    82.6  831.77
    87.5  830.85    97.2  831.32    97.6  831.39   106.9  832.97   116.6  835.11
   126.4  837.34   136.1  839.52   145.8  841.62   155.5  843.75   165.2  845.89
     175  848.03   184.7  850.45   194.4  853.24   204.1  856.42   213.8  859.71
   223.6  862.97
#Mann= 3 , 0 , 0
       0      .1       0    82.6    .045       0    97.6      .1       0
Bank Sta=82.6,97.6
XS Rating Curve= 0 ,0
Exp/Cntr=0.3,0.1

Type RM Length L Ch R = 1 ,9205.4  ,197.7,196,193.5
XS GIS Cut Line= 3
     1666327.856      647358.895     1666276.858      647388.192
     1666172.692      647476.083
#Sta/Elev= 23
       0  845.65     9.8  843.86    19.6   842.1    29.4  840.36    39.2   838.6
      49  836.78    58.8  834.63    68.6  831.96    78.3  829.17    85.2   828.1
      88  827.67    97.8  827.78   100.2  828.09   107.5  829.04   117.2  832.19
     127  836.38   136.7  840.94   146.4  845.59   156.2  850.32   165.9  854.85
   175.6  858.98   185.4  862.58   195.1  865.79
#Mann= 3 , 0 , 0
       0      .1       0    85.2    .045       0   100.2      .1       0
Bank Sta=85.2,100.2
XS Rating Curve= 0 ,0
Exp/Cntr=0.3,0.1

Type RM Length L Ch R = 1 ,9009.5  ,138.1,138.5,138.9
XS GIS Cut Line= 3
     1666213.924      647193.965     1666165.096      647235.197
     1666053.334      647348.045
#Sta/Elev= 27
       0  854.71     9.1   851.4    18.3  848.21    27.4  845.08    36.5  841.98
    45.6  838.89    54.8  835.59    63.9  831.92    73.2  827.46    80.3  825.04
    82.6  824.26    91.9  823.47    95.3  823.99   101.3  824.91   110.6  826.74
     120  828.54   129.3  829.93   138.6  831.86     148  834.43   157.3  837.18
   166.7   839.8     176  842.33   185.4  844.73   194.7  847.15     204  849.64
   213.4  852.25   222.7  854.97
#Mann= 3 , 0 , 0
       0      .1       0    80.3    .045       0   101.3      .1       0
Bank Sta=80.3,101.3
XS Rating Curve= 0 ,0
Exp/Cntr=0.3,0.1

Type RM Length L Ch R = 1 ,8871    ,285.9,277.4,268.1
XS GIS Cut Line= 4
     1666085.886      647119.095     1666064.185      647141.881
     1665987.145      647216.751     1665956.763      647279.685
#Sta/Elev= 26
       0  843.33     7.9   839.2    15.7  835.07    23.6  830.82    31.5  825.66
    41.2  819.42    44.5  818.13      51   815.6    59.5  816.22    60.8  816.31
    70.5  817.71    80.3     819    90.1  819.91    99.8  820.75   109.6  821.58
   119.4  822.23   129.1  822.95   138.9  824.49   147.6   827.5   156.4     831
   165.1  834.44   173.8  837.77   182.6  841.03   191.3   844.4     200  848.01
   208.8  851.77
#Mann= 3 , 0 , 0
       0      .1       0    44.5    .045       0    60.8      .1       0
Bank Sta=44.5,60.8
XS Rating Curve= 0 ,0
Exp/Cntr=0.3,0.1

Type RM Length L Ch R = 1 ,8593.6  ,144.9,166.7,188.1
XS GIS Cut Line= 4
     1665828.725      646983.461     1665814.619      647020.354
     1665796.172      647062.671     1665785.322      647148.392
#Sta/Elev= 22
       0  819.82     7.9  819.65    15.8  819.42    23.7  819.16    31.6  818.72
    39.5  817.86    48.7  815.79    56.9  813.11      58  812.75    67.2  812.44
    71.9   814.1    76.4  815.68    85.7  821.39    95.3  827.49   104.9  833.19
   114.5  838.53   124.1  843.54   133.7     848   143.3  852.49   152.9  857.06
   162.5  861.61   172.1  866.05
#Mann= 3 , 0 , 0
       0      .1       0    56.9    .045       0    71.9      .1       0
Bank Sta=56.9,71.9
XS Rating Curve= 0 ,0
Exp/Cntr=0.3,0.1

Type RM Length L Ch R = 1 ,8426.9  ,60.8,78.6,95.8
XS GIS Cut Line= 3
     1665770.131      646903.166     1665737.579      646904.251
     1665625.817      646928.123
#Sta/Elev= 20
       0  817.66     8.1  816.88    16.3  816.12    24.4  815.22    32.6  813.74
    42.1  810.73   47.62808.8125    51.6  807.43    52.6  807.41    61.1  807.26
    67.6  810.52    70.7  812.08    80.2  819.71    89.7  826.85    99.2  831.42
   108.8  834.13   118.3  835.42   127.8  836.39   137.3  837.45   146.8  838.57
#Mann= 3 , 0 , 0
       0      .1       0   47.62    .045       0    67.6      .1       0
Bank Sta=47.62,67.6
XS Rating Curve= 0 ,0
Exp/Cntr=0.3,0.1

Type RM Length L Ch R = 1 ,8348.3  ,69.6,69.4,73.7
XS GIS Cut Line= 2
     1665788.577      646881.465     1665541.181      646744.746
#Sta/Elev= 26
       0  818.58     9.8   817.7    19.5  817.02      39  816.39    58.5  815.29
    68.2   814.3      78  811.81    87.7  807.41    93.8  806.15    97.5  805.38
   107.2  805.31     117  806.13   126.7  807.21   136.5  808.57   146.2  809.16
     156  810.16   165.7  810.54   175.4  811.64   185.2  812.27   204.7  813.86
   214.4  815.29   224.2  816.04   243.7  818.36   263.2  820.39   272.9   822.2
   282.7  824.27
#Mann= 3 , 0 , 0
       0     .06       0    93.8    .045       0     117      .1       0
#XS Ineff= 2 , 0
       0                     137       0     815
Permanent Ineff=
       F       F
Bank Sta=93.8,117
XS Rating Curve= 0 ,0
Exp/Cntr=0.3,0.1

Type RM Length L Ch R = 1 ,8278.9  ,124.7,110.3,92
XS GIS Cut Line= 2
     1665801.598      646820.701     1665554.202      646683.982
#Sta/Elev= 23
       0  818.83      39     814    48.7  812.58    58.5  811.27      78  809.05
    87.7  807.76   107.2  804.21     117   803.2   126.4  803.51   126.7  803.52
   136.5  805.57   146.2  808.64     156   810.9   165.7  812.06   175.4  812.84
   194.9     814   204.7  814.45   224.2  815.58   233.9  816.19   243.7  816.97
   263.2  819.86   272.9  821.48   282.7  822.95
#Mann= 3 , 0 , 0
       0     .06       0   107.2    .045       0   126.4      .1       0
Bank Sta=107.2,126.4
XS Rating Curve= 0 ,0
Exp/Cntr=0.3,0.1

Type RM Length L Ch R = 1 ,8168.7  ,96.9,89.5,82.3
XS GIS Cut Line= 5
     1665866.702      646702.428      1665765.79      646646.005
     1665747.344        646653.6     1665583.499      646669.876
      1665528.16      646667.706
#Sta/Elev= 30
       0  862.15    19.3  852.48    28.9  849.42    48.2  847.84    57.8   846.1
    67.4  843.68    77.1  841.05    96.4  834.82     106     832   115.6  829.68
   128.9  821.86   135.6  818.03   145.2  813.87   154.9  811.16   164.6  809.94
   174.3  809.44   193.7  808.75   203.4  807.92     213  806.04   223.1  803.68
   232.4  802.85   242.1  803.88   251.8  805.79   261.5  807.82   271.2  809.65
   290.5  813.48   318.7  819.31   337.1  823.42   346.4  825.35   355.6  826.95
#Mann= 3 , 0 , 0
       0      .1       0   223.1    .045       0   242.1      .1       0
Bank Sta=223.1,242.1
XS Rating Curve= 0 ,0
Exp/Cntr=0.3,0.1

Type RM Length L Ch R = 1 ,8079.2  ,53.3,82.4,107.9
XS GIS Cut Line= 4
     1665652.943      646562.454     1665636.667       646574.39
     1665590.009      646592.836     1665515.139      646618.878
#Sta/Elev= 21
       0  827.13     6.7  823.41    13.5  819.28    20.2  814.59    28.6  808.72
    33.5  806.26    36.9  804.55    45.3  803.38    48.5  804.66    53.6  806.69
      62  811.48    70.4  815.22    79.2   817.2      88  817.87    96.8   818.1
   105.6  818.61   114.4   819.3   123.2  820.24     132  821.72   140.8  823.84
   149.6  826.35
#Mann= 3 , 0 , 0
       0      .1       0    33.5    .045       0    48.5      .1       0
Bank Sta=33.5,48.5
XS Rating Curve= 0 ,0
Exp/Cntr=0.3,0.1

Type RM Length L Ch R = 1 ,7996.9  ,222.8,219.3,222.1
XS GIS Cut Line= 3
     1665705.027      646585.241     1665624.731      646504.946
     1665508.629      646408.374
#Sta/Elev= 27
       0  835.39     9.5  835.87    18.9   836.1    28.4  836.09    37.8  836.23
    56.8  837.32    66.2  835.71    75.7  831.42    85.2  824.01    94.6  815.56
   104.1  808.11  109.74805.3652   113.6  803.49     123  804.23   128.1  806.03
   132.4  807.55   141.9  812.45   151.3  819.33   160.8  827.03   170.2  833.45
   179.6   836.6   189.1   837.7   217.4   841.8   226.8  843.08   236.2  844.01
   255.1  845.53   264.6  846.45
#Mann= 3 , 0 , 0
       0      .1       0  109.74    .045       0   128.1      .1       0
Bank Sta=109.74,128.1
XS Rating Curve= 0 ,0
Exp/Cntr=0.3,0.1

Type RM Length L Ch R = 1 ,7777.5  ,165.9,140.5,110.5
XS GIS Cut Line= 3
     1665762.535      646385.588      1665682.24      646305.293
     1665566.138      646208.722
#Sta/Elev= 24
       0  830.93    37.8  818.57    47.3  815.71    56.8  812.67    66.2  810.04
    75.7  807.73    85.2  805.06    94.6  803.21   104.1  801.47   113.6  799.08
     123  796.01   132.4  793.45   136.5  792.89   141.9  792.15   151.3  792.34
   151.5  792.42   160.8  796.17   170.2  800.85   179.6  803.53   189.1  805.04
   198.5  805.63   207.9  806.09   236.2  807.18   264.6  808.16
#Mann= 3 , 0 , 0
       0      .1       0   136.5    .045       0   151.5      .1       0
Bank Sta=136.5,151.5
XS Rating Curve= 0 ,0
Exp/Cntr=0.3,0.1

Type RM Length L Ch R = 1 ,7637    ,121.4,121.1,120.5
XS GIS Cut Line= 2
     1665681.155      646125.171     1665548.777      646183.765
#Sta/Elev= 18
       0  815.21     9.6  809.71    19.3  804.41      29  800.16    38.6  796.67
    48.3  792.96    57.9  788.98    65.5  786.81    67.6  786.21    77.2  786.21
    80.5  787.18    86.9  789.05    96.5  792.54   106.2  793.86   115.8  794.59
   125.5  795.74   135.1   798.2   144.8  803.06
#Mann= 3 , 0 , 0
       0      .1       0    65.5    .045       0    80.5      .1       0
Bank Sta=65.5,80.5
XS Rating Curve= 0 ,0
Exp/Cntr=0.3,0.1

Type RM Length L Ch R = 1 ,7516    ,145.7,144.6,143.4
XS GIS Cut Line= 3
     1665621.476       646032.94     1665580.244      646037.281
     1665496.693      646076.343
#Sta/Elev= 18
       0  800.87     8.3  798.83    16.6  796.84    24.9  794.92    33.2  792.88
    41.5  790.46    50.7  787.32    59.2   784.8    59.9  784.59    69.1  783.84
    74.2  784.31    78.4   784.7    87.6  788.01    96.8  792.95     106  796.94
   115.2  799.69   124.5  804.08   133.7  811.93
#Mann= 3 , 0 , 0
       0      .1       0    59.2    .045       0    78.4      .1       0
Bank Sta=59.2,78.4
XS Rating Curve= 0 ,0
Exp/Cntr=0.3,0.1

Type RM Length L Ch R = 1 ,7371.4  ,155.4,143.9,131.4
XS GIS Cut Line= 3
     1665572.648      645887.541     1665536.841      645898.392
      1665444.61       645947.22
#Sta/Elev= 18
       0  797.12     9.4  793.95    18.7  792.14    28.1  790.58    37.4  788.31
    46.9  784.65    56.4   780.3    62.1  778.61    65.9  777.48    75.4  777.86
    77.1  778.59    84.8   781.9    94.3  787.06   103.8  790.58   113.3  793.41
   122.8  796.27   132.3  799.54   141.8   803.3
#Mann= 3 , 0 , 0
       0      .1       0    62.1    .045       0    77.1      .1       0
Bank Sta=62.1,77.1
XS Rating Curve= 0 ,0
Exp/Cntr=0.3,0.1

Type RM Length L Ch R = 1 ,7227.5  ,148.3,158.8,168.5
XS GIS Cut Line= 3
     1665459.801      645748.652     1665437.014      645775.779
      1665371.91      645879.946
#Sta/Elev= 20
       0  785.18     8.9  780.83    17.7  778.58    26.6  778.12    35.4  777.81
    44.9  775.42    54.3  771.69    62.2  769.16    63.8  768.65    73.2  767.37
    77.2     768    82.7  768.86    92.1  771.71   101.6  775.32     111  779.78
   120.5  785.65   129.9     792   139.4  797.99   148.8  803.17   158.3  807.07
#Mann= 3 , 0 , 0
       0      .1       0    62.2    .045       0    82.7      .1       0
Bank Sta=62.2,82.7
XS Rating Curve= 0 ,0
Exp/Cntr=0.3,0.1

Type RM Length L Ch R = 1 ,7068.6  ,180.2,181.2,181.9
XS GIS Cut Line= 3
      1665371.91      645668.357     1665321.997      645695.484
     1665238.447      645748.652
#Sta/Elev= 21
       0   777.7     9.5  774.14    18.9  772.71    28.4  772.64    37.9  772.69
    47.3  772.77    56.8  771.68    65.8  769.78    74.8  767.28   79.93765.8585
    83.1  764.98    83.8  764.79    92.8  764.42    98.1   766.7   101.8   768.3
   110.8  775.74   119.8   783.7   128.8  790.11   137.8  796.08   146.8  801.99
   155.8  807.83
#Mann= 3 , 0 , 0
       0      .1       0   79.93    .045       0    98.1      .1       0
Bank Sta=79.93,98.1
XS Rating Curve= 0 ,0
Exp/Cntr=0.3,0.1

Type RM Length L Ch R = 1 ,6887.5  ,84.7,84.7,84.5
XS GIS Cut Line= 4
      1665290.53      645525.128     1665236.277      645539.234
     1665185.278      645569.616      1665136.45      645621.699
#Sta/Elev= 24
       0  777.65     9.3  773.18    18.7  770.53      28  769.37    37.4  768.63
    46.7  767.88    56.1     767    64.5  765.83      73   764.2    74.1  763.99
    81.5  762.54    89.1  762.56      90  762.56    98.5  764.32   106.9  767.61
   115.4  770.79   124.3   773.5   133.3  775.65   142.2  777.74   151.1  780.48
     160  784.32     169  789.51   177.9  795.26   186.8  800.48
#Mann= 3 , 0 , 0
       0      .1       0    74.1    .045       0      90      .1       0
Bank Sta=74.1,90
XS Rating Curve= 0 ,0
Exp/Cntr=0.3,0.1

Type RM Length L Ch R = 1 ,6802.8  ,88.5,89.8,90.6
XS GIS Cut Line= 3
     1665256.893      645439.407      1665213.49      645462.194
     1665065.921      645542.489
#Sta/Elev= 26
       0  775.27     9.8  770.53    19.6  766.51    29.4  764.18    39.2  764.16
      49  764.65    58.4  764.34    67.7  763.06      77  761.47    78.4  761.34
    86.4  760.57    93.4  761.07    95.7  761.24     105  762.15   114.4  762.87
   123.7  763.44     133  764.15   142.4     766   151.7  769.64     161   773.7
   170.4   777.8   179.7  781.85     189   786.2   198.4  791.69   207.7  798.73
     217  806.53
#Mann= 3 , 0 , 0
       0      .1       0      77    .045       0    95.7      .1       0
#XS Ineff= 2 , 0
       0      49     770               0
Permanent Ineff=
       F       F
Bank Sta=77,95.7
XS Rating Curve= 0 ,0
Exp/Cntr=0.3,0.1

Type RM Length L Ch R = 1 ,6713    ,195.4,214.7,218.7
XS GIS Cut Line= 3
     1665237.362      645355.857     1665195.044      645374.303
     1665031.198      645462.194
#Sta/Elev= 27
       0  786.75     9.2  781.78    18.5  776.88    27.7  772.15    36.9   767.7
    46.2  764.34      56  762.65    65.7  761.97    75.5     761    84.3  759.64
    85.3  759.48    95.1  758.95    99.3  759.07   104.9  759.22   114.7   759.7
   124.4  760.19   134.2  760.62     144  761.26   153.8  762.79   163.6  765.66
   173.4  769.17   183.2  772.69     193  776.27   202.7  780.35   212.5  786.18
   222.3  794.41   232.1   803.8
#Mann= 3 , 0 , 0
       0      .1       0    84.3    .045       0   104.9      .1       0
Bank Sta=84.3,104.9
XS Rating Curve= 0 ,0
Exp/Cntr=0.3,0.1

Type RM Length L Ch R = 1 ,6498.3  ,197.1,191,197.1
XS GIS Cut Line= 4
     1665175.513      645184.416      1665134.28      645214.798
     1665006.242      645279.902     1664954.159      645302.689
#Sta/Elev= 30
       0  777.17     8.5  773.74    17.1  770.39    25.6  767.39    34.1     765
    42.7  763.24    51.2  761.92    60.8  760.68    70.4  759.74      80  759.02
    89.5  758.32    99.1  757.73   102.2  757.69   108.7  757.62   117.2  757.68
   118.2  757.69   127.8  757.98   137.4  758.33     147  758.64   156.6   758.9
   166.1  759.11   175.7  759.31   185.3  761.04   194.9  766.92   204.3  775.21
   213.8  783.66   223.3  791.59   232.8  799.72   242.2  807.86   251.7  815.41
#Mann= 3 , 0 , 0
       0      .1       0    99.1    .045       0   118.2      .1       0
Bank Sta=99.1,118.2
XS Rating Curve= 0 ,0
Exp/Cntr=0.3,0.1

Type RM Length L Ch R = 1 ,6307.3  ,135.4,133.5,128.7
XS GIS Cut Line= 3
     1665152.726      645127.993     1665089.792      645120.397
     1664941.138      645106.291
#Sta/Elev= 26
       0  775.41     9.1  771.84    18.1  768.28    27.2  764.85    36.2  762.12
    45.3  760.48    54.3  759.51    63.4  758.56    72.7  757.51    82.1  756.35
    91.4  754.96   100.7  753.59   102.4  753.46     110  752.86   117.4  753.31
   119.4  753.43   128.7  754.47     138  755.82   147.4  758.74   156.7  763.61
     166  769.46   175.4  775.71   184.7  781.78     194  786.43   203.4  788.93
   212.7  790.37
#Mann= 3 , 0 , 0
       0      .1       0   102.4    .045       0   119.4      .1       0
Bank Sta=102.4,119.4
XS Rating Curve= 0 ,0
Exp/Cntr=0.3,0.1

Type RM Length L Ch R = 1 ,6173.8  ,188.9,168.9,148.5
XS GIS Cut Line= 2
      1665209.15      645006.465     1664951.988      644996.699
#Sta/Elev= 30
       0  834.03     9.5  828.92    19.1  823.71    28.6  818.36    38.1  812.84
    47.7  807.14    57.2  801.31    66.7  795.32    76.2  789.39    85.8  783.86
    95.3  778.68   104.8  773.56   114.4  768.24   123.9  761.92   133.4  755.23
   141.4  751.43     143  750.67   152.5  749.38   156.4   749.5     162  749.67
   171.6  750.41   181.1  751.38   190.6  752.36   200.2   753.3   209.7  754.19
   219.2  755.12   228.8  756.26   238.3  758.36   247.8   763.1   257.4  770.48
#Mann= 3 , 0 , 0
       0      .1       0   141.4    .045       0     162      .1       0
Bank Sta=141.4,162
XS Rating Curve= 0 ,0
Exp/Cntr=0.3,0.1

Type RM Length L Ch R = 1 ,6004.9  ,128.8,126.7,124.8
XS GIS Cut Line= 3
     1665089.792        644778.6     1665012.752        644851.3
     1664909.671      644957.637
#Sta/Elev= 30
       0   834.9     9.6   832.5    19.3  829.52    28.9  825.61    38.5  821.14
    48.2  815.72    57.8  809.14    67.4  801.11      77  791.25    86.7   780.6
    96.3  769.64   105.9  758.03   115.2  749.36   120.7  746.82   124.4  745.11
   133.7  744.89   135.7  745.18     143  746.22   152.2  747.78   161.5  749.27
   170.7   750.6     180  751.75   189.2  752.82   198.5   753.6   207.7  754.12
     217  754.41   226.3  755.25   235.5  757.66   244.8  762.26     254  767.28
#Mann= 3 , 0 , 0
       0      .1       0   120.7    .045       0     143      .1       0
Bank Sta=120.7,143
XS Rating Curve= 0 ,0
Exp/Cntr=0.3,0.1

Type RM Length L Ch R = 1 ,5878.2  ,104,103.5,103.1
XS GIS Cut Line= 3
     1664943.308      644730.857     1664916.181      644768.835
     1664846.737      644854.555
#Sta/Elev= 20
       0  772.87     9.3  768.26    18.7  763.94      28  760.02    37.3  756.17
    46.7  752.15    55.9  747.39    65.1  743.21    67.2  742.95    74.2   742.1
    82.2  743.59    83.4  743.81    92.6  747.58   101.8  751.77     111  755.73
   120.2  758.92   129.4  761.21   138.6  762.07   147.8  762.68     157   763.1
#Mann= 3 , 0 , 0
       0      .1       0    65.1    .045       0    83.4      .1       0
Bank Sta=65.1,83.4
XS Rating Curve= 0 ,0
Exp/Cntr=0.3,0.1

Type RM Length L Ch R = 1 ,5774.7  ,253,239.1,222.2
XS GIS Cut Line= 3
      1664898.82      644594.138     1664836.971       644703.73
     1664770.782      644786.196
#Sta/Elev= 27
       0  814.17     9.7  809.14    19.4  803.57      29  798.14    38.7  792.13
    48.4  786.26    58.1  780.16    67.8  774.39    77.4  768.82    87.1  763.55
    96.8  759.24   106.5  755.65   116.2  752.16   125.8  748.06   135.4  743.92
     137  743.59   145.1  741.94     152     743   154.7  743.42   164.3   746.3
   173.9  749.56   183.5  753.25   193.1  757.21   202.7  760.59   212.4  761.84
     222  762.28   231.6  762.47
#Mann= 3 , 0 , 0
       0      .1       0     137    .045       0   154.7      .1       0
Bank Sta=137,154.7
XS Rating Curve= 0 ,0
Exp/Cntr=0.3,0.1

Type RM Length L Ch R = 1 ,5535.7  ,258.5,270,281.8
XS GIS Cut Line= 3
     1664651.424      644487.802     1664639.488      644614.755
     1664640.573      644767.749
#Sta/Elev= 25
       0  840.49     9.8     833    19.6  825.39    58.8  794.57    68.7  786.92
    78.5  779.58    88.3  772.56    98.1   765.7   107.9     759   117.7  752.79
   127.5  746.77   137.1  741.67   146.6  738.72   156.2  737.99   165.8  738.65
   175.3  740.02   184.9  742.67   194.4  747.73     204  754.25   213.6  759.16
   223.1  760.95   232.7  761.13   251.8  761.27   261.4  761.45   280.5  761.96
#Mann= 3 , 0 , 0
       0      .1       0   146.6    .045       0   165.8      .1       0
Bank Sta=146.6,165.8
XS Rating Curve= 0 ,0
Exp/Cntr=0.3,0.1

Type RM Length L Ch R = 1 ,5265.7  ,153.1,153,152.7
XS GIS Cut Line= 3
      1664423.56       644534.46     1664402.943      644563.756
     1664325.903       644697.22
#Sta/Elev= 23
       0  773.09       9  766.41    17.9  759.38    26.9   752.1    35.8  745.72
    45.5  741.03    55.1  738.56    64.7  737.15    74.4  735.96    74.5  735.96
      84  735.94    89.5  737.22    93.6  738.18   103.2  743.53   112.9   749.2
   122.5  751.95   132.1  753.16   141.8  754.13   151.4  755.09     161  756.08
   170.7  757.06   180.3  758.06   189.9   759.3
#Mann= 3 , 0 , 0
       0      .1       0    74.4    .045       0    89.5      .1       0
Bank Sta=74.4,89.5
XS Rating Curve= 0 ,0
Exp/Cntr=0.3,0.1

Type RM Length L Ch R = 1 ,5112.7  ,153.7,157.4,161.2
XS GIS Cut Line= 3
     1664292.266       644463.93      1664267.31      644494.312
     1664202.205      644609.329
#Sta/Elev= 21
       0  762.83     9.8  755.14    19.7  749.07    29.5  744.34    39.3   740.6
    48.8  737.96    58.2  736.44    67.6  735.55    77.1   734.7    80.2  734.57
    86.5   734.3    95.2  734.93      96  734.99   105.4  737.52   114.8  741.25
   124.3   744.7   133.7  747.29   143.2  749.43   152.6  751.45     162  753.44
   171.5  755.45
#Mann= 3 , 0 , 0
       0      .1       0    77.1    .045       0      96      .1       0
Bank Sta=77.1,96
XS Rating Curve= 0 ,0
Exp/Cntr=0.3,0.1

Type RM Length L Ch R = 1 ,4955.3  ,131.1,131.4,131.3
XS GIS Cut Line= 3
     1664169.653       644386.89     1664138.186      644418.357
      1664047.04      644531.204
#Sta/Elev= 23
       0  753.03     8.9  749.18    17.8  745.53    26.7  742.07    35.6  739.15
    44.5  736.92    54.2   735.4    63.8  734.42    73.5  733.43    82.3  732.44
    83.2  732.34    92.8  731.31    97.3  732.07   102.5  732.94   112.2  736.81
   121.9  741.82   131.5  745.24   141.2  748.19   150.9  750.92   160.6  753.58
   170.2  756.34   179.9  759.34   189.6  763.72
#Mann= 3 , 0 , 0
       0      .1       0    82.3    .045       0   102.5      .1       0
Bank Sta=82.3,102.5
XS Rating Curve= 0 ,0
Exp/Cntr=0.3,0.1

Type RM Length L Ch R = 1 ,4823.8  ,129.5,137.4,145.4
XS GIS Cut Line= 3
     1664064.402      644308.765      1664034.02      644339.147
     1663948.299      644444.399
#Sta/Elev= 22
       0  744.73     8.6  739.86    17.2  736.63    25.8  735.38    34.4  734.79
      43  733.96    52.7   732.8    62.4   731.2      72  729.54    75.5  729.19
    81.8  728.57    90.5  730.29    91.4  730.47   101.1  734.48   110.8  739.17
   120.5  742.23   130.2  744.22   139.9  745.88   149.6  747.48   159.3  749.48
     169  752.61   178.7  755.69
#Mann= 3 , 0 , 0
       0      .1       0      72    .045       0    91.4      .1       0
Bank Sta=72,91.4
XS Rating Curve= 0 ,0
Exp/Cntr=0.3,0.1

Type RM Length L Ch R = 1 ,4686.5  ,221.7,234.9,247.3
XS GIS Cut Line= 4
     1664003.638      644216.534      1663959.15      644242.576
     1663902.726      644276.213     1663850.643      644327.211
#Sta/Elev= 24
       0  748.14     8.6  744.88    17.2  741.38    25.8  737.79    34.4  734.49
      43  731.66    51.6  729.34    60.9  726.73    68.4   725.2    70.3  724.81
    79.7  724.49    83.4   724.7    89.1  725.03    98.5  726.02   107.8  727.83
   117.2  730.97   126.4  734.36   135.5  737.86   144.6  741.18   153.7  744.12
   162.8  746.68   171.9  749.16     181  751.71   190.1  754.26
#Mann= 3 , 0 , 0
       0      .1       0    68.4    .045       0    89.1      .1       0
Bank Sta=68.4,89.1
XS Rating Curve= 0 ,0
Exp/Cntr=0.3,0.1

Type RM Length L Ch R = 1 ,4451.5  ,98.7,91.4,83
XS GIS Cut Line= 3
     1663924.428      644066.795     1663872.344      644080.901
     1663697.648       644078.73
#Sta/Elev= 27
       0  734.61       9  732.61      18  731.41      27  730.53      36  729.66
      45  728.81      54  727.98    63.7  727.13    73.4  726.29    83.1  725.48
    92.8  724.68   102.5  723.85   112.2  722.83   119.8  721.91   121.9  721.66
   131.6  720.92   134.8   721.4   141.3  722.37     151  727.43   160.7  733.87
   170.4  739.62   180.1  744.31   189.8  748.24   199.6  751.84   209.3  755.46
     219  759.11   228.7  762.82
#Mann= 3 , 0 , 0
       0      .1       0   119.8    .045       0   141.3      .1       0
Bank Sta=119.8,141.3
XS Rating Curve= 0 ,0
Exp/Cntr=0.3,0.1

Type RM Length L Ch R = 1 ,4360.2  ,88.5,96.1,102.8
XS GIS Cut Line= 3
     1663898.386      643975.649     1663848.473      643973.479
     1663726.945      644014.711
#Sta/Elev= 22
       0  728.16     8.3  727.53    16.6  726.96      25   726.4    33.3  725.81
    41.6  725.14      50  724.38    59.1   723.7    68.3   722.8    77.5  721.62
    86.6     720    95.7  718.55     105  718.63   110.7  720.16   114.1  721.07
   123.3     725   132.5  728.87   141.6  732.32   150.8  735.66     160  738.98
   169.1  742.48   178.3  746.15
#Mann= 3 , 0 , 0
       0      .1       0    86.6    .045       0   110.7      .1       0
Bank Sta=86.6,110.7
XS Rating Curve= 0 ,0
Exp/Cntr=0.3,0.1

Type RM Length L Ch R = 1 ,4264.1  ,231.8,222.2,211.6
XS GIS Cut Line= 4
     1663899.471      643904.034     1663840.877      643900.779
     1663749.731      643900.779     1663704.159      643917.055
#Sta/Elev= 24
       0  733.73     9.8  730.63    19.6  728.02    29.3     726    39.1  724.28
    48.9  722.82    58.7  721.52    67.8   720.4    76.9  719.24      86   717.9
    95.1  716.96    96.9   716.9   104.3  716.64   111.9  717.37   113.4  717.51
   122.5  719.88   131.6  722.98   140.7  725.96   149.8  728.61   159.5  731.38
   169.2  734.17   178.9  736.88   188.5  739.61   198.2  742.48
#Mann= 3 , 0 , 0
       0      .1       0    95.1    .045       0   113.4      .1       0
Bank Sta=95.1,113.4
XS Rating Curve= 0 ,0
Exp/Cntr=0.3,0.1

Type RM Length L Ch R = 1 ,4041.9  ,148.2,145,140.9
XS GIS Cut Line= 3
     1663821.346      643658.808     1663782.284       643687.02
     1663652.075      643751.039
#Sta/Elev= 23
       0  736.89     9.6  730.14    19.3  726.23    28.9  724.48    38.6  723.38
    48.2  721.33    57.9  718.23    67.5  715.19    68.2  715.11    77.2  714.07
    83.2  714.42    86.9  714.63    96.6  715.86   106.2  717.09   115.9  718.15
   125.6  719.14   135.2  720.16   144.9   721.2   154.6  722.22   164.3  723.24
   173.9  724.32   183.6  725.66   193.3  728.04
#Mann= 3 , 0 , 0
       0      .1       0    68.2    .045       0    86.9      .1       0
Bank Sta=68.2,86.9
XS Rating Curve= 0 ,0
Exp/Cntr=0.3,0.1

Type RM Length L Ch R = 1 ,3896.9  ,97.1,101.6,105.7
XS GIS Cut Line= 4
     1663756.242      643535.111      1663723.69      643549.216
     1663657.501       643596.96     1663577.205      643656.638
#Sta/Elev= 27
       0  724.48     8.9  721.76    17.7  719.62    26.6  717.88    35.5  716.24
    44.5  714.38    53.6  712.34    62.7  710.49    68.1  709.89    71.8  709.48
    80.8  710.04    83.1  710.44    89.9  711.62      99  713.39     108  714.95
   117.1  716.15   126.2  717.36   135.3  718.59   144.4  719.91   153.5  721.34
   162.6  722.95   171.7  724.72   180.8  726.86   189.8  729.68   198.9  733.02
     208  736.77   217.1  740.92
#Mann= 3 , 0 , 0
       0      .1       0    62.7    .045       0    83.1      .1       0
Bank Sta=62.7,83.1
XS Rating Curve= 0 ,0
Exp/Cntr=0.3,0.1

Type RM Length L Ch R = 1 ,3795.3  ,131.6,138.2,144.3
XS GIS Cut Line= 3
     1663703.073      643470.006     1663659.671      643487.368
     1663527.292      643550.302
#Sta/Elev= 23
       0   719.9     9.4  718.28    18.7  716.93      28   715.6    37.4   714.4
    46.8  713.15    56.5  711.99    66.3  710.86    76.1  709.61    85.8  708.41
    92.8  707.58    95.6  707.25   105.4  706.95   107.8  707.42   115.2  708.87
   124.9  713.02   134.7  717.91   144.5  722.42   154.2  726.42     164  729.48
   173.8   731.5   183.6  732.61   193.3  734.15
#Mann= 3 , 0 , 0
       0      .1       0    92.8    .045       0   107.8      .1       0
Bank Sta=92.8,107.8
XS Rating Curve= 0 ,0
Exp/Cntr=0.3,0.1

Type RM Length L Ch R = 1 ,3657.2  ,183.1,175.2,166.8
XS GIS Cut Line= 4
      1663655.33      643361.499     1663623.863       643374.52
     1663535.973      643387.541     1663462.188      643419.008
#Sta/Elev= 27
       0  723.45     8.5  717.94      17  714.79    25.5  713.31      34  712.34
    42.9   711.5    51.8  710.63    60.7  709.57    69.6  708.24    78.5  706.68
   83.48705.9803    86.4  705.57    87.4  705.43    96.2  705.13   101.4  705.92
   105.1  706.48     114  709.61   122.9  713.34   131.8  716.52   140.7  719.56
   149.6  722.61   158.6  725.34   167.5   727.4   176.4   728.7   185.3  729.71
   194.2  730.95   203.1  732.71
#Mann= 3 , 0 , 0
       0      .1       0   83.48    .045       0   101.4      .1       0
Bank Sta=83.48,101.4
XS Rating Curve= 0 ,0
Exp/Cntr=0.3,0.1

Type RM Length L Ch R = 1 ,3482    ,212.2,216.8,220.7
XS GIS Cut Line= 4
      1663569.61      643186.803     1663538.143      643203.079
     1663477.379      643236.716     1663420.955      643260.588
#Sta/Elev= 22
       0  732.15     8.9  726.54    17.7   721.5    26.6  716.91    35.4  712.76
    44.1   709.1    52.8   705.9    60.5  704.14    61.5  703.91    70.2  703.48
    75.5  704.29    78.8  704.79    87.5  707.67    96.2  711.06   104.9  714.15
   113.6  716.93   122.4  719.67   131.1  722.52   139.9  725.39   148.6  728.26
   157.4  731.01   166.2  732.92
#Mann= 3 , 0 , 0
       0      .1       0    60.5    .045       0    78.8      .1       0
Bank Sta=60.5,78.8
XS Rating Curve= 0 ,0
Exp/Cntr=0.3,0.1

Type RM Length L Ch R = 1 ,3265.2  ,123.5,114.6,105
XS GIS Cut Line= 4
     1663484.975      643006.682     1663436.146      643025.128
     1663350.426       643053.34     1663296.172      643089.147
#Sta/Elev= 26
       0  736.29     8.7  731.22    17.4  726.28    26.1  721.55    34.8  716.95
    43.5  712.68    52.2  708.94    61.2  705.41    70.2  702.02    79.3  699.92
    80.3  699.85    88.3  699.31    95.3  699.63    97.3  699.72   106.3  700.75
   115.4  702.02   124.4  703.26   133.4  704.57   142.4  706.49   151.7  709.64
     161  713.31   170.3  717.16   179.6  721.09   188.9  725.03   198.2  728.86
   207.4  732.57
#Mann= 3 , 0 , 0
       0      .1       0    79.3    .045       0    97.3      .1       0
Bank Sta=79.3,97.3
XS Rating Curve= 0 ,0
Exp/Cntr=0.3,0.1

Type RM Length L Ch R = 1 ,3150.5  ,99.6,98.4,96.5
XS GIS Cut Line= 4
     1663398.169      642904.685     1663364.532      642928.557
     1663309.193       642978.47     1663274.471      643029.468
#Sta/Elev= 23
       0   713.2     8.2  710.47    16.5  708.12    24.8  706.61      33  705.74
    41.2     704    50.6   701.7    59.9  699.48    61.7  699.37    69.2   698.9
    76.7  699.23    78.5  699.31    87.8  700.43    97.1  701.61   106.4  702.63
   115.8  703.53   124.6  704.46   133.4  705.59   142.2  707.67     151  710.64
   159.8  714.25   168.6  718.33   177.5   722.7
#Mann= 3 , 0 , 0
       0      .1       0    59.9    .045       0    78.5      .1       0
Bank Sta=59.9,78.5
XS Rating Curve= 0 ,0
Exp/Cntr=0.3,0.1

Type RM Length L Ch R = 1 ,3052.2  ,168.8,170,169.2
XS GIS Cut Line= 4
     1663359.106       642822.22     1663304.853      642851.517
     1663219.132      642937.237     1663183.325      643000.171
#Sta/Elev= 27
       0  724.36     8.8  719.83    17.6   714.9    26.4   710.3    35.2  706.93
      44   704.9    52.8  703.51    61.7  702.28      71  701.26    80.3  700.44
      99  698.14   108.3  697.17   117.6  697.56   121.8  698.01   136.3  699.54
   154.9  700.33   164.2     701   173.6  702.22   182.9  703.87   191.9  705.96
     201  708.52     210  711.69   219.1  715.46   228.1  719.83   237.2  724.64
   246.2  729.89   255.3  735.35
#Mann= 3 , 0 , 0
       0      .1       0      99    .045       0   121.8      .1       0
Bank Sta=99,121.8
XS Rating Curve= 0 ,0
Exp/Cntr=0.3,0.1

Type RM Length L Ch R = 1 ,2882.1  ,135.1,148.3,160
XS GIS Cut Line= 4
     1663240.834      642711.543     1663201.771      642739.755
      1663096.52      642853.687     1663045.521      642925.302
#Sta/Elev= 23
       0  706.76     9.6  705.16    28.9   703.4    38.6  702.34    48.2  700.25
    57.9  697.08      65  695.59    67.6  695.05    77.3  694.82      87  695.32
    96.7  695.79   135.4   697.2   154.8  697.78   183.9   698.5   193.6  698.86
   203.3   699.9   213.1  703.24   222.8  708.36   232.6  714.29   242.4  720.55
   261.9   733.3   281.4  745.74   291.2  751.83
#Mann= 3 , 0 , 0
       0      .1       0      65    .045       0      87      .1       0
Bank Sta=65,87
XS Rating Curve= 0 ,0
Exp/Cntr=0.3,0.1

Type RM Length L Ch R = 1 ,2733.8  ,140.3,128.6,116.2
XS GIS Cut Line= 4
     1663185.495      642609.546     1663117.136      642652.949
     1663008.629      642686.586     1662905.547       642826.56
#Sta/Elev= 28
       0  716.17       9  713.89      36   706.8      45  704.32      54  702.02
      63  700.36      81  698.28    90.4  696.97    99.9  694.95   108.5  693.28
   109.4   693.1   118.8  692.67   128.3  693.77   137.8  695.75   147.2  696.87
   156.7  697.06   175.6  696.82   185.1  696.79   194.6  696.89   213.9  697.34
   242.9  698.23   281.5  699.65   291.2  700.55   300.8  703.57   310.5  708.42
   329.8  719.33   349.1  730.96   368.4  742.81
#Mann= 3 , 0 , 0
       0      .1       0   108.5    .045       0   128.3      .1       0
Bank Sta=108.5,128.3
XS Rating Curve= 0 ,0
Exp/Cntr=0.3,0.1

Type RM Length L Ch R = 1 ,2605.2  ,173.4,163.2,150.4
XS GIS Cut Line= 4
     1663068.308       642509.72     1663048.777      642530.336
     1662971.737      642614.972      1662871.91      642780.987
#Sta/Elev= 23
       0  721.54    18.9  711.13    28.4  705.47    37.9     699    47.5  693.69
      57  691.46    57.7  691.43    66.6   691.1    76.1  691.55   114.2  694.22
   133.3  695.45   142.8  695.96   152.5  696.35   191.3  697.28   220.3  698.22
   249.4  699.28   268.8  699.77   278.4   700.3   288.1  702.22   297.8   706.1
   307.5  710.57   326.9  718.82   336.6  723.31
#Mann= 3 , 0 , 0
       0      .1       0    57.7    .045       0    76.1      .1       0
Bank Sta=57.7,76.1
XS Rating Curve= 0 ,0
Exp/Cntr=0.3,0.1

Type RM Length L Ch R = 1 ,2442    ,159.2,160.8,161.2
XS GIS Cut Line= 4
     1662905.547      642443.531     1662889.271      642480.423
     1662845.869      642613.887     1662782.935      642678.991
#Sta/Elev= 24
       0  722.07     8.1  716.96    16.1   712.2    24.2  707.57    32.3  702.82
    40.3  697.76    49.7  692.04    56.9  689.22      59   688.4    68.4  687.49
    77.8  688.02    96.5   689.9   124.5  692.34   133.9  693.09   143.2  693.65
     162  694.39   171.3  694.97   180.7  695.78   189.7  697.03   198.8  699.69
     244  715.61   253.1  718.45   262.2  720.85   271.2  722.98
#Mann= 3 , 0 , 0
       0      .1       0    56.9    .045       0    77.8      .1       0
Bank Sta=56.9,77.8
XS Rating Curve= 0 ,0
Exp/Cntr=0.3,0.1

Type RM Length L Ch R = 1 ,2281.1  ,80.6,72.9,65
XS GIS Cut Line= 4
     1662765.573      642419.659     1662748.212      642461.977
     1662721.086      642541.187      1662711.32      642604.121
#Sta/Elev= 24
       0  700.06     9.2  698.01    18.3   696.1    27.4  694.36    36.6   692.7
    45.7  691.09      55   689.6    64.4  688.15    73.6   686.6      83  684.95
    89.3  684.28    92.3  683.96   101.6  684.17   104.3  684.84   110.9  686.49
   120.2  690.89   129.5  695.93   138.6  700.11   147.7  704.06   156.8  708.09
   165.9   712.2     175   716.2   184.1   719.8   193.2  722.74
#Mann= 3 , 0 , 0
       0      .1       0      83    .045       0   104.3      .1       0
Bank Sta=83,104.3
XS Rating Curve= 0 ,0
Exp/Cntr=0.3,0.1

Type RM Length L Ch R = 1 ,2208.2  ,153.8,145,135.9
XS GIS Cut Line= 4
     1662645.131      642392.532     1662660.322      642444.616
     1662661.407      642523.826     1662657.067      642600.866
#Sta/Elev= 26
       0  715.32       9  710.01    18.1  705.04    27.1  700.36    36.2  696.18
    45.2  692.78    54.2  690.27    63.1  688.49    71.9  687.15    80.7  685.99
    89.5  684.84    95.8   684.2    98.3  683.94   107.1  683.71   110.8  684.29
   115.9   685.1   124.7   688.3   133.5  692.44   143.1  696.88   152.8  701.04
   162.4  705.16     172  709.26   181.7  713.31   191.3  717.25     201  721.06
   210.6  724.52
#Mann= 3 , 0 , 0
       0      .1       0    95.8    .045       0   115.9      .1       0
Bank Sta=95.8,115.9
XS Rating Curve= 0 ,0
Exp/Cntr=0.3,0.1

Type RM Length L Ch R = 1 ,2063.2  ,144.4,140.8,136
XS GIS Cut Line= 2
     1662486.711       642426.17     1662553.985       642582.42
#Sta/Elev= 22
       0  723.68     9.4   717.6    18.9   711.3    28.4  704.85    37.8  698.59
    47.2  692.99    56.7   688.6    66.2  685.18    71.8  684.02    75.6  683.24
    85.1  683.17    86.8  683.51   88.96683.9392    94.5  685.04     104   688.5
   113.4  692.22   122.9  695.46   132.3  698.57   141.8  701.65   151.2  704.74
   160.7  707.83   170.1  710.87
#Mann= 3 , 0 , 0
       0      .1       0    71.8    .045       0   88.96      .1       0
Bank Sta=71.8,88.96
XS Rating Curve= 0 ,0
Exp/Cntr=0.3,0.1

Type RM Length L Ch R = 1 ,1922.5  ,127.9,120.3,112.5
XS GIS Cut Line= 4
     1662372.778      642518.401     1662386.884      642553.123
     1662417.266      642597.611     1662451.988      642634.503
#Sta/Elev= 19
       0  707.12     9.4  701.96    18.7   696.6    28.1     691    37.5   685.3
    46.5   680.8    50.5  679.96    55.4  678.94    64.4  679.76    65.5  680.03
    73.4     682    82.4  684.91    91.4  687.58    99.8   689.9   108.2  692.22
   116.7   694.6   125.1  697.03   133.6  699.45     142  701.91
#Mann= 3 , 0 , 0
       0      .1       0    46.5    .045       0    65.5      .1       0
Bank Sta=46.5,65.5
XS Rating Curve= 0 ,0
Exp/Cntr=0.3,0.1

Type RM Length L Ch R = 1 ,1802.2  ,201.8,207.2,212.4
XS GIS Cut Line= 4
     1662259.931      642621.482     1662293.568      642639.928
     1662352.162      642683.331      1662396.65      642721.308
#Sta/Elev= 21
       0  702.45     9.6  697.41    19.2  692.51    28.8  687.89    38.4  683.24
    47.5  679.06    54.5     677    56.6  676.38    65.7  675.95    69.5  676.55
    74.8  677.38    83.9  679.84      93  682.44   102.2  684.93   111.3  687.39
     121  690.04   130.8  692.66   140.5  695.26   150.3  697.74     160  699.94
   169.8  702.04
#Mann= 3 , 0 , 0
       0      .1       0    54.5    .045       0    69.5      .1       0
Bank Sta=54.5,69.5
XS Rating Curve= 0 ,0
Exp/Cntr=0.3,0.1

Type RM Length L Ch R = 1 ,1595    ,77.3,82.2,86.1
XS GIS Cut Line= 4
     1662137.318      642750.605      1662161.19      642790.753
     1662195.912      642831.986     1662232.804      642878.644
#Sta/Elev= 22
       0  712.57     9.3  707.97    18.7  702.88      28  696.69    37.4  689.59
    46.7  681.68    55.7  675.32   60.58673.8698    62.8  673.21    64.7  672.64
    73.7  673.11    77.8  674.31    82.6  675.72    91.6  679.46   100.6   683.1
   109.1   686.5   117.6  689.89   126.1  693.22   134.6  696.51   143.1  699.69
   151.6  702.59   160.1  705.45
#Mann= 3 , 0 , 0
       0      .1       0   60.58    .045       0    77.8      .1       0
Bank Sta=60.58,77.8
XS Rating Curve= 0 ,0
Exp/Cntr=0.3,0.1

Type RM Length L Ch R = 1 ,1512.7  ,130.7,126.4,121.6
XS GIS Cut Line= 4
     1662076.554      642790.753      1662088.49       642815.71
     1662123.212      642878.644     1662178.551      642945.918
#Sta/Elev= 23
       0  707.34     9.2  701.02    18.4  693.03    27.7  683.29    36.6  675.01
    41.9  672.99    45.6  671.58    54.6  671.33    56.9  671.73    63.6  672.89
    72.6  675.17    81.6  677.26    90.6  678.97    99.5  680.21   109.2  681.19
   118.9  682.13   128.6  683.58   138.3  685.63   147.9  688.02   157.6  690.73
   167.3  694.07     177  697.72   186.6  701.54
#Mann= 3 , 0 , 0
       0      .1       0    41.9    .045       0    63.6      .1       0
Bank Sta=41.9,63.6
XS Rating Curve= 0 ,0
Exp/Cntr=0.3,0.1

Type RM Length L Ch R = 1 ,1386.3  ,154.5,171.7,188
XS GIS Cut Line= 4
     1661965.877      642861.282     1661979.983      642886.239
     1662048.343      642966.534      1662081.98      643041.404
#Sta/Elev= 26
       0  702.85     9.6  696.47    19.1  688.92    28.7  680.52    38.2  672.53
    44.1  669.78    47.8  668.06    57.4  667.79    59.1  668.03      67  669.17
    76.6  671.18    86.2  672.69    95.8   673.8   105.4  674.51     115  675.06
   124.5   675.5   134.1  676.11   143.2  676.83   152.4  678.18   161.5  680.22
   170.6  682.99   179.7  686.12   188.8  689.43     198  693.02   207.1  696.72
   216.2  700.55
#Mann= 3 , 0 , 0
       0      .1       0    44.1    .045       0      67      .1       0
Bank Sta=44.1,67
XS Rating Curve= 0 ,0
Exp/Cntr=0.3,0.1

Type RM Length L Ch R = 1 ,1214.6  ,98.5,119.5,139.5
XS GIS Cut Line= 4
     1661881.242      642911.196      1661857.37      642966.534
     1661854.115       643059.85     1661901.858      643184.633
#Sta/Elev= 28
       0     688     8.6  685.14    17.2  682.42    25.8   679.9    34.4  678.21
      43  677.07    51.7  675.67    60.3  673.95    69.6  670.75    78.9  666.39
    81.7  665.57    88.3  663.63    97.6  664.38   116.3  671.04   125.6  672.93
     135  674.19   153.6   675.9   163.2  677.26   182.3  680.61   191.8  682.39
   201.4  684.38   220.4   688.8     230  690.56   239.5  691.35   249.1  691.47
   258.6  691.96   268.2     693   287.2  695.25
#Mann= 3 , 0 , 0
       0      .1       0    81.7    .045       0    97.6      .1       0
Bank Sta=81.7,97.6
XS Rating Curve= 0 ,0
Exp/Cntr=0.3,0.1

Type RM Length L Ch R = 1 ,1095.1  ,116.8,133.7,149.6
XS GIS Cut Line= 4
     1661851.945      642875.388     1661815.053      642891.664
     1661732.587      642952.428     1661628.421      643043.574
#Sta/Elev= 27
       0   688.4     8.1  684.26    16.1  679.82    24.2  675.62    32.3  671.81
    40.3  668.54    49.6  666.21      59  664.45    68.3  662.97    77.6  661.65
    86.9  660.86    96.2  661.01    98.6  661.48   105.5  662.85   114.8  665.86
   124.1  669.08   133.4     672   179.7  686.06   188.9  688.97   198.1  692.02
   207.4  694.74   216.6  696.71   225.8  697.77   253.5  700.36   262.7  701.54
   271.9  703.62   281.2  706.31
#Mann= 3 , 0 , 0
       0      .1       0    77.6    .045       0    98.6      .1       0
Bank Sta=77.6,98.6
XS Rating Curve= 0 ,0
Exp/Cntr=0.3,0.1

Type RM Length L Ch R = 1 ,961.4   ,140.6,122.4,104.1
XS GIS Cut Line= 4
     1661806.372      642795.093     1661765.139      642807.029
     1661679.419      642799.433     1661642.527      642816.795
#Sta/Elev= 22
       0  686.37     8.6  681.36    17.2   676.3    25.8  671.65    34.3  668.06
    42.9  665.93    52.5  664.04      62  661.74    71.6  659.08    76.5  658.31
    81.2  657.58    90.7  658.63    91.5  658.92   100.3  662.08   109.9  666.34
   119.4  669.61     129  672.12   137.1   673.3   145.3  674.46   153.4  675.78
   161.6  677.69   169.8  680.16
#Mann= 3 , 0 , 0
       0      .1       0    71.6    .045       0    90.7      .1       0
Bank Sta=71.6,90.7
XS Rating Curve= 0 ,0
Exp/Cntr=0.3,0.1

Type RM Length L Ch R = 1 ,839     ,220.6,189,156.4
XS GIS Cut Line= 4
     1661760.799      642649.694     1661743.438       642665.97
     1661691.355      642710.458     1661630.591      642808.114
#Sta/Elev= 25
       0  705.29     7.9  701.94    15.9  697.16    23.8   689.1    33.6  673.71
    43.4  660.96    48.8  658.86    53.2  657.14    62.9  657.95    63.8   658.2
    72.7  660.64    82.5  662.56    92.3   663.9   101.9   664.9   111.5  665.69
     121  666.39   130.6  667.08   140.2   667.9   149.8  668.85   159.4  669.84
     169  670.65   178.6  672.44   188.1  675.48   197.7  678.77   207.3  682.12
#Mann= 3 , 0 , 0
       0      .1       0    48.8    .045       0    63.8      .1       0
Bank Sta=48.8,63.8
XS Rating Curve= 0 ,0
Exp/Cntr=0.3,0.1

Type RM Length L Ch R = 1 ,650     ,146.4,155.9,156.3
XS GIS Cut Line= 4
     1661525.339      642578.079     1661529.679      642606.291
     1661595.869      642721.308     1661599.124      642787.498
#Sta/Elev= 27
       0  690.47     9.5  682.83      19  673.76    28.5  663.12      38  655.21
    47.5  651.64    48.7  651.56      57  650.97    63.7  651.08    66.5  651.13
    75.9   651.6    85.4  652.02    94.9  652.74   104.4  653.82   113.8  655.33
   123.3  657.16   132.8   658.9   142.3  660.66   151.8  662.24   161.2   663.7
   170.7   664.9   180.2  666.09   189.6  667.74   199.1  670.49   208.6  674.05
     218  677.58   227.5  680.94
#Mann= 3 , 0 , 0
       0      .1       0    48.7    .045       0    66.5      .1       0
Bank Sta=48.7,66.5
XS Rating Curve= 0 ,0
Exp/Cntr=0.3,0.1

Type RM Length L Ch R = 1 ,494.1   ,181.3,212,243.4
XS GIS Cut Line= 5
      1661463.49      642578.079     1661458.065      642652.949
      1661465.66      642697.437     1661516.543      642767.409
     1661515.675      642868.972
#Sta/Elev= 30
       0  696.54     9.4  694.26    18.8  691.02    37.5  683.61    56.3  676.49
    75.1  668.75    84.1  666.08    93.1  663.83   102.2  661.86   111.2  660.21
   129.8  657.33   139.4  654.78     149  652.57   158.6  650.68   168.3  649.89
   177.9  649.45   187.5  649.44   194.6   651.9   197.1  652.77   206.7  661.34
     216  673.91   225.2  687.06   234.4  696.82   243.6  702.98   252.9  706.51
   262.1  708.71   271.4  710.12   280.6  710.92   289.8  711.31   308.3  711.69
#Mann= 3 , 0 , 0
       0      .1       0   177.9    .045       0   194.6      .1       0
Bank Sta=177.9,194.6
XS Rating Curve= 0 ,0
Exp/Cntr=0.3,0.1

Type RM Length L Ch R = 1 ,282.1   ,192.1,182.4,173
XS GIS Cut Line= 4
     1661455.895      642559.633     1661400.556      642594.355
     1661352.813      642635.588      1661298.56      642696.352
#Sta/Elev= 26
       0  697.08     9.3  692.74    18.7  687.82      28  682.45    37.3   676.7
    46.7  670.83      56  664.93    65.3  658.76    74.3     653    83.4  649.41
    88.9  648.48    92.4  647.88   101.4   647.9   103.9  648.35   110.4  649.52
   119.4  652.39   128.4  656.03   137.5  659.71   146.5  663.55   155.6  667.46
   164.6  671.77   173.7  676.41   182.7  681.68   191.8  687.26   200.8  692.88
   209.9  698.39
#Mann= 3 , 0 , 0
       0      .1       0    88.9    .045       0   103.9      .1       0
Bank Sta=88.9,103.9
XS Rating Curve= 0 ,0
Exp/Cntr=0.3,0.1
